--- MILLCREEK1.prj (project) ---

Proj Title=MILLCREEK1
Current Plan=p01
Default Exp/Contr=0,0
English Units
Geom File=g01
Flow File=f01
Plan File=p01
BEGIN DESCRIPTION:
END DESCRIPTION:
DSS Export Rating Curves= 0
DSS Export Rating Curve Sorted= 0
DSS Export Volume Flow Curves= 0
DXF OffsetX= 0
DXF OffsetY= 0
DXF ScaleX= 0
DXF ScaleY= 0

--- MILLCREEK1.p01 (plan) ---

Plan Title=Floodplain
Program Version=4.00
Geom File=g01
Flow File=f01
K Sum by GR=0
Std Step Tol=0.01
Critical Tol=0.01
Num of Std Step Trials=20
Max Error Tol=0.3
Flow Tol Ratio=0.001
Split Flow NTrial=30
Split Flow Tol=0.02
Split Flow Ratio=0.02
Log Output Level=0
Friction Slope Method=1
Unsteady Friction Slope Method=2
Unsteady Bridges Friction Slope Method=1
Global Log Level=0
CheckData=False
Run HTab=0
Run UNet=0
Run PostProcess=0
UNET Theta=0
UNET Theta Warmup=0
UNET ZTol=0
UNET ZSATol=0
UNET MxIter=0
UNET MaxInSteps=0
UNET DtIC=0
UNET DtMin=0
UNET MaxCRTS=0
UNET WFStab=0
UNET SFStab=0
UNET WFX=0
UNET SFX=0
UNET DSS MLevel=0
UNET DZMax Abort=0
UNET Convert EG Bridges=0
UNET Use Existing IB Tables=0
UNET Froude Limit=0
UNET Froude Power=0
Write IC File=0
Echo Input=False
Echo Output=False
Write Detailed=0

--- MILLCREEK1.f01 (steady flow) ---

Flow Title=NFF Regression Equation
Program Version=4.10
Number of Profiles= 1
Profile Names=P100yr
River Rch & RM=MILLCREEK1,Main            ,17670.2
 541.236
River Rch & RM=MILLCREEK1,Main            ,16112.4
600.4815
River Rch & RM=MILLCREEK1,Main            ,15787.6
 681.103
River Rch & RM=MILLCREEK1,Main            ,14712.1
753.3466
River Rch & RM=MILLCREEK1,Main            ,13817
  813.59
River Rch & RM=MILLCREEK1,Main            ,12212.3
887.8899
River Rch & RM=MILLCREEK1,Main            ,11052.9
926.2821
River Rch & RM=MILLCREEK1,Main            ,7933.3
1001.352
River Rch & RM=MILLCREEK1,Main            ,7362.8
1183.885
River Rch & RM=MILLCREEK1,Main            ,211.4
1292.034
Boundary for River Rch & Prof#=MILLCREEK1,Main            , 1
Up Type= 0
Dn Type= 1
Dn Known WS=660.5
DSS Import GetInterval= 0
DSS Import GetPeak= 0
DSS Import FillOption= 0

--- MILLCREEK1.g01 (geometry) ---

Geom Title=USGS 10m DEM
Program Version=5.03

River Reach=MILLCREEK1      ,Main
Reach XY= 30
     2356043.593      307760.166      2356147.76      308614.333
     2356823.392      309684.127     2357222.446      310020.895
     2357678.614      310078.987     2358826.091       310942.51
     2358970.528      311194.022     2359724.149      311310.513
      2360033.24      311486.276     2360123.132      311709.647
     2359970.676      312124.749     2360743.246       312642.11
     2360829.825      312888.502     2360717.204      313050.096
     2361163.384      313246.277     2361396.522      313686.667
     2361989.774      313713.291     2362149.578      314113.298
     2362353.653      314126.522      2362342.72      314272.152
     2362842.204      314603.916     2363215.468      315161.207
     2363514.079      315284.471     2363550.537      315584.819
     2363801.569      315950.481     2363704.955      316485.377
     2364259.121      317495.272      2364145.58      318095.012
      2364345.24       318397.38     2364286.649      318840.027

Type RM Length L Ch R = 1 ,17670.2 ,411.5,423.8,396.7
XS GIS Cut Line= 3
      2355656.75      307894.454     2356046.641       307769.69
     2356429.887      307623.285
#Sta/Elev= 30
       0  751.89   50.19752.3196    55.6  752.12    59.6  750.23    63.6  747.36
    67.6  746.13    87.4  745.53   96.15  751.44    99.4  751.83     147   749.5
   222.6  742.97   282.2  734.76     306  729.91   325.9  727.15   357.7  725.43
   397.4  725.58   405.4  724.36   413.4  723.15   421.3  724.38   445.2  725.43
   508.9  726.08   544.8   728.5   576.7  728.19   600.6   728.9   628.4     733
   648.4  734.43   684.2  738.72   763.9  751.61   791.7  754.75   819.6  756.73
#Mann= 5 ,-1 , 0
       0     .12       0   50.19    .016       0   96.15     .12       0
   405.4    .045       0   421.3     .12       0
Bank Sta=405.4,421.3
XS Rating Curve= 0 ,0
Exp/Cntr=0.3,0.1

Type RM Length L Ch R = 1 ,17246.4 ,141.4,146.1,158.2
XS GIS Cut Line= 3
     2355689.243      308161.982     2355927.958      308113.154
     2356514.981      308110.984
#Sta/Elev= 30
       0  742.53      28  741.02    63.9   738.1   123.8  735.05  193.18733.2932
   203.7  731.08   219.7  731.02  236.93729.8416   267.6  726.32   283.6  725.27
   303.6  725.29   327.5  724.21   367.4  723.62   399.4  724.39   403.4  723.18
   407.4   722.3   419.4  723.34   431.4  724.34   455.3   723.4   479.3  723.47
   511.2  725.32   539.2  728.74   563.1  733.31   587.1  740.28     639  749.22
   710.9  757.85  763.43761.1131   790.8  762.38   824.2 762.535   830.7  762.43
#Mann= 7 ,-1 , 0
       0     .12       0  193.18    .016       0  236.93     .12       0
   403.4    .045       0   419.4     .12       0  763.43     .06       0
   824.2     .12       0
Bank Sta=403.4,419.4
XS Rating Curve= 0 ,0
Exp/Cntr=0.3,0.1

Type RM Length L Ch R = 1 ,17100.3 ,101.9,102.1,102.1
XS GIS Cut Line= 4
     2355691.413       308285.68     2355982.212      308232.512
     2356230.693         308277.     2356531.257      308126.175
#Sta/Elev= 30
       0  745.29      36  742.92    59.9  739.71   115.8  735.28   148.3735.4762
   158.9735.6865  182.25735.4478   207.7  735.38   223.7  732.91   267.7  728.27
   303.5  726.42  316.58725.0208   335.1  723.71   366.6  723.48   374.5  722.37
   382.4  722.97   398.2  723.97   421.8   724.1     481  723.29   512.6  724.34
   559.9  727.29   599.5  731.94     647   741.7   670.7  745.32   686.5  746.99
   706.3  750.23  720.49749.9611  774.33754.4492   832.9   759.2   884.3  761.58
#Mann= 9 ,-1 , 0
       0     .12       0   148.3     .06       0   158.9     .12       0
  182.25    .016       0  316.58     .12       0   366.6    .045       0
   382.4     .12       0  720.49     .06       0  774.33     .12       0
#XS Ineff= 2 , 0
          347.78  725.15  401.44          725.57
Permanent Ineff=
       F       F
Bank Sta=366.6,382.4
XS Rating Curve= 0 ,0
Exp/Cntr=0.3,0.1

Type RM Length L Ch R = 1 ,16998.3 ,166.3,156.1,145.9
XS GIS Cut Line= 4
     2355702.264      308381.167     2355993.062      308327.998
     2356241.543      308372.486     2356542.108      308221.661
#Sta/Elev= 30
       0  743.32   57.26743.4634    79.9  743.06    95.9  740.72   107.9  739.91
   135.8  741.03   155.5740.7307  179.84740.0177  222.41738.0903   291.6  727.78
  321.26724.7894   370.6  722.95   382.4  720.82   390.3   720.4  395.88 720.997
   403.8722.5875  495.79 723.312   528.3  724.75     552  726.96   567.8  727.28
   578.5729.4954   619.3  735.43     639  739.44   654.9  740.86   674.6  744.82
   726.1  748.98   749.6748.4105   817.1  751.65  839.92751.8232   884.3  754.44
#Mann= 13 ,-1 , 0
       0     .12       0   57.26    .016       0   155.5     .06       0
  179.84    .016       0  222.41     .06       0  321.26     .12       0
   382.4    .045       0  395.88     .12       0   403.8     .06       0
  495.79    .016       0   578.5     .12       0   749.6     .06       0
  839.92     .12       0
#XS Ineff= 2 , 0
          356.04  724.73  436.53          724.61
Permanent Ineff=
       F       F
Bank Sta=382.4,395.88
XS Rating Curve= 0 ,0
Exp/Cntr=0.3,0.1

Type RM Length L Ch R = 1 ,16842.2 ,379,376.5,373.9
XS GIS Cut Line= 2
     2355743.496      308599.265        2356579.      308371.401
#Sta/Elev= 30
       0  752.87   38.13751.7654  192.72745.1732  221.41 742.122   251.4  739.99
  263.82737.9661   291.3  729.53   315.3  723.78   327.2  722.76   359.2  722.61
   376.2  720.91   383.1  720.02   391.2  721.18   399.1   722.3   494.9  722.14
  526.96724.1568  531.77724.7177   550.7  729.24   570.7  729.71   574.7  730.12
   580.4732.0535   594.6  735.52   618.6   737.3   646.5  741.38  660.95742.0654
   706.4  747.25   738.3  748.68  768.42752.0287   802.2  754.92     866  758.69
#Mann= 12 ,-1 , 0
       0    .016       0   38.13     .12       0  192.72     .06       0
  221.41    .016       0  263.82     .12       0   376.2    .045       0
   391.2     .12       0  526.96     .06       0  531.77    .016       0
   580.4     .06       0  660.95    .016       0  768.42     .12       0
Bank Sta=376.2,391.2
XS Rating Curve= 0 ,0
Exp/Cntr=0.3,0.1

Type RM Length L Ch R = 1 ,16465.7 ,351.5,353.4,355.5
XS GIS Cut Line= 3
     2355886.726      308990.976     2356518.236      308739.239
     2356646.274      308599.265
#Sta/Elev= 30
       0  749.11   36.73747.4117   69.33745.7735   77.99745.3308  121.08742.8687
  234.55734.6214  275.78729.5862  307.35724.8237   339.9  721.03   395.9  720.93
  405.99719.7988   411.9  718.76  421.03719.7879   479.9  721.79   487.9  720.54
   511.9  720.48   536.2 724.952   551.9   728.4  571.49730.6277   595.9  733.56
   611.8  733.25  623.06737.0534  654.63739.3767  655.55739.4894   675.8  742.82
  694.09744.0174  729.65744.3542   743.1  744.36   786.5  750.12   869.5  756.52
#Mann= 17 ,-1 , 0
       0     .06       0   36.73    .016       0   69.33     .06       0
   77.99    .016       0  121.08     .06       0  234.55    .016       0
  275.78     .06       0  307.35     .12       0  405.99    .045       0
  421.03     .12       0   536.2     .06       0  571.49    .016       0
  623.06     .12       0  654.63     .06       0  655.55     .12       0
  694.09     .08       0  729.65     .12       0
Bank Sta=405.99,421.03
XS Rating Curve= 0 ,0
Exp/Cntr=0.3,0.1

Type RM Length L Ch R = 1 ,16112.4 ,322.4,324.8,277.6
XS GIS Cut Line= 3
     2356142.802      309430.429      2356264.33      309176.522
     2356924.052      308973.614
#Sta/Elev= 30
       0  736.09   37.44734.7606   61.21733.2435   142.7  730.76   206.2  727.56
   245.8   727.1   269.6  725.48   301.4  726.05  368.83723.6017  401.33723.3561
     453  721.19     493  718.81  499.73717.5784   508.9  716.36  514.15717.5869
   520.9  719.27   548.8  718.14   600.7  721.36  616.16723.2562   632.6  727.76
   644.6  728.44   656.5  727.82     667729.8613  686.19731.6588  710.13734.4892
   788.2  740.58     868   742.6   883.9  744.49   895.9  743.89   971.7  747.29
#Mann= 11 ,-1 , 0
       0     .12       0   37.44    .016       0   61.21     .12       0
  368.83    .016       0  401.33     .12       0  499.73    .045       0
  514.15     .12       0  616.16    .016       0     667     .12       0
  686.19     .06       0  710.13     .12       0
Bank Sta=499.73,514.15
XS Rating Curve= 0 ,0
Exp/Cntr=0.3,0.1

Type RM Length L Ch R = 1 ,15787.6 ,81.3,71.8,68.8
XS GIS Cut Line= 3
     2356190.545      309503.128     2356410.814      309360.984
     2356959.859      309170.012
#Sta/Elev= 30
       0  737.89   80.95732.6747  142.65729.9589   166.8  728.63   202.6  727.83
   246.3  725.31     286  721.59     302  718.64   313.9  717.56   357.7  717.84
  367.81716.1592   377.6  715.36   382.5  716.19   401.5  718.46   413.4  717.97
   477.2  718.42  499.98  721.42   532.9  727.28  543.71728.5866   560.8   729.9
  578.77729.9839   580.7  730.23   588.6  733.58   624.5     735   684.2  740.17
  717.95742.3134   771.8   742.8   811.3744.0255  827.37744.6393   843.5  745.68
#Mann= 11 ,-1 , 0
       0     .12       0   80.95     .06       0  142.65     .12       0
  367.81    .045       0   382.5     .12       0  499.98     .06       0
  543.71    .016       0  578.77     .06       0  717.95     .12       0
   811.3     .06       0  827.37     .08       0
Bank Sta=367.81,382.5
XS Rating Curve= 0 ,0
Exp/Cntr=0.3,0.1

Type RM Length L Ch R = 1 ,15715.8 ,57.6,58.1,58.1
XS GIS Cut Line= 3
     2356267.585      309587.764     2356684.252      309275.264
     2356962.029      309181.948
#Sta/Elev= 30
       0  734.91   28.98 733.474   66.01731.3135      79730.6537  116.31727.9413
  151.89725.7042  166.62724.9609  188.34723.8762   246.5  720.99   266.4  717.06
  342.94717.9314   353.8  717.77   366.2  715.46   377.7  715.23   381.2  715.38
   393.6  717.77   425.4  718.46   449.3  720.01  476.22723.9148   517.3728.5487
   532.7  729.74  548.01729.8162   552.5  730.26   560.4  732.94   564.4  733.26
   596.1  734.32   639.6  738.05  689.39740.9398  795.76743.6135   813.9  744.74
#Mann= 16 ,-1 , 0
       0     .06       0   28.98    .016       0   66.01     .12       0
      79    .016       0  116.31     .06       0  151.89    .016       0
  166.62     .06       0  188.34    .016       0  342.94     .12       0
   366.2    .045       0   381.2     .12       0  476.22     .06       0
   517.3    .016       0  548.01     .06       0  689.39     .12       0
  795.76     .08       0
#XS Ineff= 2 , 0
          344.69  720.02  398.35          720.07
Permanent Ineff=
       F       F
Bank Sta=366.2,381.2
XS Rating Curve= 0 ,0
Exp/Cntr=0.3,0.1

Type RM Length L Ch R = 1 ,15657.7 ,174.1,176.6,170
XS GIS Cut Line= 3
     2356308.818      309623.571     2356761.292      309292.625
      2356972.88       309216.67
#Sta/Elev= 30
       0  734.99    1.08734.9657    19.9  734.12   64.71 730.949   111.3  727.13
   147.1  724.84   186.9     723   270.4  717.04   298.2     718     334  717.76
   341.9  717.49   348.1716.3406   353.8  715.19   357.8  715.43   361.8  716.28
   369.8  718.14   397.6  719.29   429.4  722.69  462.21725.5656  488.47727.3838
   508.9  729.61   528.8  729.34  534.48730.1755   548.7  731.39  614.65734.3287
  659.06736.7058  702.38739.3362  710.16739.7355   765.7  742.06   785.4  743.44
#Mann= 12 ,-1 , 0
       0    .016       0    1.08     .06       0   64.71     .12       0
   348.1    .045       0   361.8     .12       0  462.21     .06       0
  488.47    .016       0  534.48     .12       0  614.65     .06       0
  659.06     .12       0  702.38     .06       0  710.16     .12       0
#XS Ineff= 2 , 0
          317.03  719.92  375.64          719.76
Permanent Ineff=
       F       F
Bank Sta=348.1,361.8
XS Rating Curve= 0 ,0
Exp/Cntr=0.3,0.1

Type RM Length L Ch R = 1 ,15481.1 ,324.1,313.3,287.3
XS GIS Cut Line= 2
     2356404.986      309750.843     2357014.113      309276.349
#Sta/Elev= 30
       0  731.69    19.9  730.48    39.8  728.42    67.7  726.86   151.2  720.76
   218.9  717.03   230.8  716.59   258.7  717.14   282.6  716.53   298.5  716.65
   318.4  715.95   334.3   716.7  340.42715.9838   350.2   715.3  355.68715.9087
   366.2  717.48   386.1  718.22   449.7   726.8   465.7  728.74  471.99728.7104
   501.5  728.32  502.59728.8078   505.5  730.11   509.4  732.69   513.4  733.97
   535.6735.1665   628.8  743.82  672.85746.2375   688.6   745.5   772.1  745.79
#Mann= 7 ,-1 , 0
       0     .12       0  340.42    .045       0  355.68     .12       0
  471.99    .016       0  502.59     .12       0   535.6     .06       0
  672.85     .08       0
Bank Sta=340.42,355.68
XS Rating Curve= 0 ,0
Exp/Cntr=0.3,0.1

Type RM Length L Ch R = 1 ,15167.9 ,318.3,321.8,319.5
XS GIS Cut Line= 3
      2356739.59      309979.474     2356984.816      309491.193
     2357095.493      309362.069
#Sta/Elev= 30
       0  720.13   119.6  718.14   127.6  717.54   167.5  716.74   187.4  716.72
   223.4  715.19   271.2  714.81   287.2  715.54   305.1  714.18   311.1  712.87
   315.1  713.09   320.1  714.84     327  716.25   362.9   717.6  390.63722.7393
   398.8  725.45   406.8  726.53   426.8   725.7  429.46 726.041   430.7   726.2
   438.7  731.56   442.7  732.67   466.6  734.42   502.5  738.29   530.4   740.6
   613.6  749.42   657.1   752.3   676.9  752.48   714.2754.1695   716.5  754.25
#Mann= 6 ,-1 , 0
       0     .12       0   305.1    .045       0   320.1     .12       0
  390.63    .016       0  429.46     .12       0   714.2     .06       0
Bank Sta=305.1,320.1
XS Rating Curve= 0 ,0
Exp/Cntr=0.3,0.1

Type RM Length L Ch R = 1 ,14846.1 ,85.5,86.2,85.9
XS GIS Cut Line= 2
     2356978.305      310086.896     2357320.102      309492.278
#Sta/Elev= 30
       0  722.39    23.9  721.26    71.8  717.97   103.7  714.89   147.5  714.16
   191.4  714.74   203.7  712.65   211.3  711.78   215.3  711.82   218.7  712.64
   227.3  714.38   231.3  714.62   263.2  715.12   291.1  714.99     315  715.94
     335  717.76  344.37 719.412  386.68728.7317   406.7  729.36   422.7  728.84
   438.2 732.287   474.5  738.09   510.4  741.05   554.3  746.66  571.26748.2328
  597.14750.2924  605.64750.9178  640.01752.7956  646.03753.1816   685.8  754.93
#Mann= 11 ,-1 , 0
       0     .12       0   203.7    .045       0   218.7     .12       0
  344.37     .06       0  386.68    .016       0   438.2     .06       0
  571.26     .08       0  597.14     .06       0  605.64     .08       0
  640.01     .06       0  646.03     .12       0
Bank Sta=203.7,218.7
XS Rating Curve= 0 ,0
Exp/Cntr=0.3,0.1

Type RM Length L Ch R = 1 ,14759.9 ,47.7,47.7,48.5
XS GIS Cut Line= 3
     2357048.636      310116.232     2357317.374      309682.466
     2357353.938      309496.579
#Sta/Elev= 30
       0  722.05    47.8  720.38    59.8  718.16    63.8  717.83   103.6  716.67
   135.5  714.44   155.5  714.58   163.4  714.18   173.8  712.21   183.4  711.66
   188.8  712.26   199.3  714.58   255.1  714.09  292.98714.8802     303   715.3
   334.9  719.49   362.8  724.27  382.41728.1752  408.79728.5169  442.21 729.082
   450.5  729.81   458.4   731.5   474.4  733.88   498.3  736.59     534  739.73
   553.7  742.15   585.3  747.84  634.25752.0172   672.1  754.44   699.7  754.77
#Mann= 8 ,-1 , 0
       0     .12       0   173.8    .045       0   188.8     .12       0
  292.98     .06       0  382.41     .08       0  408.79    .016       0
  442.21     .06       0  634.25     .12       0
Bank Sta=173.8,188.8
XS Rating Curve= 0 ,0
Exp/Cntr=0.3,0.1

Type RM Length L Ch R = 1 ,14712.1 ,77,76.2,81.7
XS GIS Cut Line= 3
     2357093.124      310134.678     2357361.861      309700.913
     2357398.426      309515.025
#Sta/Elev= 30
       0  721.46    87.7  718.88   143.5     713   151.5  712.71  157.89711.5747
   163.4  710.87  173.07711.4439   183.4  713.41  194.13 714.023  286.72713.9594
     307  714.59   346.8  718.32   370.7  724.28   386.7     729   390.7  729.34
   396.5  728.55   402.6  727.29   434.5  727.19  439.59728.6104   446.5   733.5
   450.5  735.53   454.5  736.03   474.4  736.34   518.2  738.76   537.9     741
   581.3  747.47   624.7   751.3  653.86752.6512  665.52  753.15   699.7  753.74
#Mann= 9 ,-1 , 0
       0     .12       0  157.89    .045       0  173.07     .12       0
  194.13     .06       0  286.72     .12       0   396.5    .016       0
  439.59     .06       0  653.86     .12       0  665.52     .06       0
Bank Sta=157.89,173.07
XS Rating Curve= 0 ,0
Exp/Cntr=0.3,0.1

Type RM Length L Ch R = 1 ,14636   ,228.1,227.6,220.6
XS GIS Cut Line= 3
     2357173.618      310172.616     2357416.674      309676.739
     2357448.141      309530.255
#Sta/Elev= 30
       0  721.18   85.38717.2612   123.2   715.6     147  713.34     155  713.44
   162.9   711.5   170.8  710.72  176.94711.4708   182.8  712.53   206.6  713.16
   242.4   713.5   270.2  711.72     286  713.52   317.8  713.28  335.84716.6857
   357.6  719.12  385.51 724.945   401.3  728.32   409.2  726.56  418.65726.5809
     437  726.13  441.76727.0828   448.9  733.26   452.9  735.27   456.9  736.01
   476.8  737.23   496.6  740.74   567.4745.5154   642.9  750.62   702.1  752.89
#Mann= 9 ,-1 , 0
       0     .06       0   85.38     .12       0   162.9    .045       0
  176.94     .12       0  335.84     .06       0  385.51     .08       0
  418.65    .016       0  441.76     .12       0   567.4     .06       0
Bank Sta=162.9,176.94
XS Rating Curve= 0 ,0
Exp/Cntr=0.3,0.1

Type RM Length L Ch R = 1 ,14408.4 ,266.5,271.4,275.6
XS GIS Cut Line= 3
     2357348.314      310222.529      2357514.33      309882.903
     2357583.774      309584.509
#Sta/Elev= 30
       0  719.55    71.6  717.46   111.4  715.29   117.3 715.428   123.4  715.89
   143.2  713.67  185.64 712.937   210.9  712.04   226.8  712.52   236.4  711.74
   242.7  710.78   251.4   711.6   266.6  713.04   322.3  712.42   334.3  711.65
   338.2  712.27   346.2  715.12   354.2  716.56     378  718.52  395.17 721.154
   409.9   722.6   429.8   722.6  431.53724.4142   433.7  726.69   437.7  729.13
   461.6  732.39   501.4  735.35     577  743.54  615.15745.7527   684.4  749.54
#Mann= 8 ,-1 , 0
       0     .12       0   117.3     .06       0  185.64     .12       0
   236.4    .045       0   251.4     .12       0  395.17    .016       0
  431.53     .12       0  615.15     .06       0
Bank Sta=236.4,251.4
XS Rating Curve= 0 ,0
Exp/Cntr=0.3,0.1

Type RM Length L Ch R = 1 ,14137   ,314.3,320,321.9
XS GIS Cut Line= 3
     2357507.819      310301.739     2357809.469      309903.519
     2357787.767      309655.038
#Sta/Elev= 30
       0  721.94      12  720.84      32  721.11      48  718.71    83.9   716.7
  120.72715.8705   131.9  715.08   159.9  714.15  183.19712.4549   191.8   711.7
   203.8  711.34   255.8  711.27   272.2  710.27   279.8  709.61   287.2  710.65
  308.84711.0857   331.7   711.4  399.25713.7952   423.6  715.26   435.6  715.15
  443.04716.2452   451.6   717.8   459.6  718.45   479.6  718.65   499.6  719.72
   535.2  722.83   602.5  727.23   638.1  729.35   725.2  733.62     749  735.93
#Mann= 8 ,-1 , 0
       0     .12       0  120.72     .06       0  183.19     .12       0
   272.2    .045       0   287.2     .12       0  308.84     .06       0
  399.25    .016       0  443.04     .12       0
Bank Sta=272.2,287.2
XS Rating Curve= 0 ,0
Exp/Cntr=0.3,0.1

Type RM Length L Ch R = 1 ,13817   ,50.4,50.9,51.3
XS GIS Cut Line= 2
     2357717.238      310404.821     2358207.689      309956.687
#Sta/Elev= 30
       0  724.32    31.8  721.78    43.8  723.52    47.7  723.22    59.7  719.98
   71.67719.0954    83.5  718.11   115.4  713.81   171.1   710.3  183.93709.9837
  190.75709.8456   222.8  709.41   232.8  708.51   238.7  707.97   247.8  708.62
   262.6  708.83   270.5  709.53   338.1  710.62  350.11711.2109     366  712.45
   381.9  711.68  394.03 712.522   417.7  712.72   457.5  711.94   477.4  712.64
   493.3  711.94   533.1  712.72     541  713.42   584.8   714.5   664.4  714.95
#Mann= 9 ,-1 , 0
       0     .12       0   71.67     .06       0    83.5     .12       0
  183.93     .06       0  190.75     .12       0   232.8    .045       0
   247.8     .12       0  350.11    .016       0  394.03     .12       0
Bank Sta=232.8,247.8
XS Rating Curve= 0 ,0
Exp/Cntr=0.3,0.1

Type RM Length L Ch R = 1 ,13766   ,44.4,44.4,44.3
XS GIS Cut Line= 3
     2357713.983      310426.522     2357857.212      310342.972
     2358267.368      309978.389
#Sta/Elev= 30
       0  725.53    15.8  725.31    27.6  723.81   92.58718.7466  101.77718.5222
   142.1  716.66     154   715.7   181.7  711.86   201.6  710.02   237.4  709.04
  243.93707.9047   249.3  707.38   257.3  707.85  271.97708.4485   285.1  708.27
   344.8  709.87   360.7  709.78   376.6  710.72   392.5  712.44   408.4  711.61
   427.9 712.043  428.52  712.04     472  712.39  563.56714.4806  583.88714.8961
  608.83715.2789     647  715.82   682.8  717.66  709.29717.4896   714.6  717.41
#Mann= 12 ,-1 , 0
       0     .12       0   92.58     .08       0  101.77     .12       0
  243.93    .045       0   257.3     .12       0  271.97    .016       0
   427.9     .12       0  428.52     .06       0  563.56     .08       0
  583.88     .06       0  608.83     .12       0  709.29     .06       0
Bank Sta=243.93,257.3
XS Rating Curve= 0 ,0
Exp/Cntr=0.3,0.1

Type RM Length L Ch R = 1 ,13721.7 ,94,93.9,93.9
XS GIS Cut Line= 3
     2357742.194      310459.075     2357885.424      310375.524
      2358295.58      310010.941
#Sta/Elev= 30
       0  726.16   17.54724.7827   39.42 723.326   91.45720.1757   99.71719.7278
  129.62717.8927   161.9  714.98   169.8  714.62   209.6  709.29   221.5   708.6
   245.4   708.5   249.3  708.09   253.8  706.68   257.3  706.09   268.8  706.62
   277.2  708.46     309     708  357.92709.4067  379.34711.3255   400.4   712.6
   412.4   712.2   420.3  713.36  430.61713.3823     468  713.26   559.5   715.5
  633.84 716.568  659.47717.2357  664.16 717.431  703.08718.1348   714.6  718.22
#Mann= 15 ,-1 , 0
       0     .08       0   17.54     .06       0   39.42     .08       0
   91.45     .06       0   99.71     .12       0  129.62    .016       0
   253.8    .045       0   268.8    .016       0  357.92     .08       0
  379.34    .016       0  430.61     .06       0  633.84     .08       0
  659.47     .12       0  664.16     .08       0  703.08     .06       0
Bank Sta=253.8,268.8
XS Rating Curve= 0 ,0
Exp/Cntr=0.3,0.1

Type RM Length L Ch R = 1 ,13627.8 ,204.1,205.5,202.9
XS GIS Cut Line= 2
     2357869.147      310524.179     2358324.877      310063.024
#Sta/Elev= 30
       0  725.39    43.8  722.46   60.63720.0379    71.6  718.37  108.83717.5627
   115.4  716.65   139.2   711.4   167.1  708.26     179  707.71   226.7  708.61
   230.7  708.26  237.57706.0686   242.6  705.26   250.6  706.04   258.5  707.68
   274.4  708.41   294.3  707.57   318.2  712.12  330.53713.2386     350  712.71
   365.9  713.01   369.9  713.27  376.78715.6184  389.82715.6091   409.7  715.32
   477.3  716.52     533  719.26   568.8  720.26   592.7  719.54   648.4  720.92
#Mann= 8 ,-1 , 0
       0     .06       0   60.63    .016       0  108.83     .12       0
  237.57    .045       0   250.6     .12       0  330.53    .016       0
  376.78     .12       0  389.82     .06       0
Bank Sta=237.57,250.6
XS Rating Curve= 0 ,0
Exp/Cntr=0.3,0.1

Type RM Length L Ch R = 1 ,13422.2 ,341.6,344.2,345.4
XS GIS Cut Line= 4
      2358070.97      310671.748     2358078.745      310599.196
      2358215.79       310432.48     2358446.404       310149.83
#Sta/Elev= 30
       0  720.19   52.67715.8835    65.3  715.61      73   714.8      85  714.88
   96.04714.0436   112.9  712.29   136.9  710.66   160.9  706.52   172.9  706.84
   188.9  708.58   216.8  706.45   236.8  707.26   256.8  705.55   264.8  704.41
  271.45 705.343   284.8  708.52   328.4  713.41  338.48 713.654   356.2  714.54
   364.1   714.3   368.1  714.68     372  715.98  379.46716.5833   391.9  716.01
   463.2  717.17   542.6  719.31   574.3  721.05   594.1  721.36   653.6   723.7
#Mann= 7 ,-1 , 0
       0     .06       0   52.67    .016       0   96.04     .12       0
   256.8    .045       0  271.45     .12       0  338.48    .016       0
  379.46     .06       0
Bank Sta=256.8,271.45
XS Rating Curve= 0 ,0
Exp/Cntr=0.3,0.1

Type RM Length L Ch R = 1 ,13078   ,298.8,297.2,295.7
XS GIS Cut Line= 2
     2358284.078      310857.295      2358705.33      310403.555
#Sta/Elev= 30
       0  725.58   31.54722.7148    47.9  720.01    63.9  719.55   75.55 717.081
    99.9  712.81   107.8  710.18   127.8  707.48   163.8  706.06   203.7  705.52
   215.7  705.87   239.7  704.05   247.7  704.72  254.33703.9226   263.6  702.82
   269.3703.8683   275.6  705.26   291.6  705.13   299.6  705.68   315.6   709.7
   327.5  711.84  358.44714.5438   379.5  716.02   391.5  715.97  403.12717.0025
   468.7  720.38  486.42 721.147  544.24724.7684  568.21725.4525   619.1  724.64
#Mann= 11 ,-1 , 0
       0     .06       0   31.54    .016       0   75.55     .12       0
  254.33    .045       0   269.3     .12       0  358.44    .016       0
  403.12     .06       0   468.7     .08       0  486.42     .06       0
  544.24     .08       0  568.21     .06       0
Bank Sta=254.33,269.3
XS Rating Curve= 0 ,0
Exp/Cntr=0.3,0.1

Type RM Length L Ch R = 1 ,12780.7 ,130.2,130.9,131.4
XS GIS Cut Line= 3
     2358518.887      311061.722     2358858.514       310646.14
     2358871.535      310538.719
#Sta/Elev= 30
       0   711.4    7.72711.3506    19.9  710.72    35.8  710.85   56.88708.7213
    71.6  707.18   85.61707.2144   115.3  707.33   143.1  706.64   198.8  703.87
   246.5  704.07   250.5  703.25   254.4  701.94   258.4  701.85   262.4  701.85
  269.44703.6247   274.3  704.44   302.2  705.02  329.37709.6481   337.9  710.98
  367.27712.8967  399.08714.0001   417.4  714.58   429.4  714.22   437.3  716.73
  444.64716.8328   512.8  717.67   552.2  719.31  628.18720.7695   644.9  721.36
#Mann= 11 ,-1 , 0
       0     .12       0    7.72    .016       0   56.88     .06       0
   85.61     .12       0   250.5    .045       0  269.44     .12       0
  329.37     .06       0  367.27     .12       0  399.08    .016       0
  444.64     .06       0  628.18     .12       0
Bank Sta=250.5,269.44
XS Rating Curve= 0 ,0
Exp/Cntr=0.3,0.1

Type RM Length L Ch R = 1 ,12649.8 ,98.9,98.1,97.3
XS GIS Cut Line= 2
      2358612.42      311140.064     2359007.385       310683.25
#Sta/Elev= 30
       0  711.69    5.27711.4873      80  709.43     116  709.36     128  708.81
  145.39706.8014     176  704.94     200  704.64     208  703.82     228  704.66
     244  703.18     268  703.11     276  702.38     284  701.46   291.9  702.36
   303.9  703.75   347.9     712   379.9  712.02  399.58712.6888   431.9  712.97
   443.9  712.52   447.9  712.62  453.86 713.814   483.9  715.24   523.9  719.17
  551.35720.9729  562.56720.7607   583.9   721.3  602.15720.0481   603.9  719.93
#Mann= 10 ,-1 , 0
       0    .016       0    5.27     .06       0  145.39     .12       0
     276    .045       0   291.9     .12       0  399.58    .016       0
  453.86     .12       0  551.35    .016       0  562.56     .12       0
  602.15     .06       0
Bank Sta=276,291.9
XS Rating Curve= 0 ,0
Exp/Cntr=0.3,0.1

Type RM Length L Ch R = 1 ,12551.7 ,96.4,92.9,89.8
XS GIS Cut Line= 2
      2358689.46      311198.875     2359089.851       310735.55
#Sta/Elev= 30
       0  710.07    35.8  707.68   49.29707.5159    75.6   707.6   89.77707.0936
   127.2  705.48   147.1  703.79   178.9  703.25   190.9  702.49   254.5  703.79
   266.4  701.67   274.4  700.94   282.3   700.4  288.87701.0683   302.2  703.85
   326.1  705.82   353.9  709.63   377.8  711.07  409.95712.1699   445.4  712.91
   457.3  712.48  459.73713.1968   469.2  715.58   481.1   716.2     505  719.38
   520.9  720.35   528.8  721.45   556.7  722.87   608.4  721.46   612.4  720.64
#Mann= 7 ,-1 , 0
       0     .06       0   49.29     .08       0   89.77     .12       0
   274.4    .045       0  288.87     .12       0  409.95    .016       0
  459.73     .12       0
Bank Sta=274.4,288.87
XS Rating Curve= 0 ,0
Exp/Cntr=0.3,0.1

Type RM Length L Ch R = 1 ,12458.8 ,226.8,246.5,243.4
XS GIS Cut Line= 2
     2358775.831      311258.988     2359119.799      310763.111
#Sta/Elev= 30
       0  710.65   11.99709.8209   48.34707.6015   68.12706.4679   86.97705.8072
   103.9  705.46   115.9  704.29   143.9  703.24   155.9  701.24   175.8   702.6
   223.8  702.94   231.8  702.79  237.31701.5726   247.8  700.59  252.75701.5505
   259.8  704.01   267.8  705.25   279.8  706.02   295.8   708.3   323.7  710.41
   371.7   711.2  422.56713.1652   431.6   713.1   443.6   713.9   459.6  713.68
  466.24715.2012   495.6  720.08   547.5  722.38   563.5  722.27   603.5  719.16
#Mann= 9 ,-1 , 0
       0     .06       0   11.99     .08       0   48.34     .12       0
   68.12     .06       0   86.97     .12       0  237.31    .045       0
  252.75     .12       0  422.56    .016       0  466.24     .12       0
Bank Sta=237.31,252.75
XS Rating Curve= 0 ,0
Exp/Cntr=0.3,0.1

Type RM Length L Ch R = 1 ,12212.3 ,242.4,246,243.8
XS GIS Cut Line= 2
     2358961.378      311338.849     2359212.029      310827.781
#Sta/Elev= 30
       0  709.24   15.67708.6763    79.6  704.81   103.5   704.5   111.5  703.46
   123.4  700.46   139.3  702.12   151.3  702.36   163.2  701.46   171.2  701.58
  184.68699.4846   191.1  698.34  199.75699.5372     207  702.53     211   703.4
   218.9  704.45   234.8  705.25   253.3707.0325   318.4  711.53   374.2   713.8
   400.5713.9684   429.9  714.82   441.8   714.7  451.81715.3298   461.8   715.6
   489.6  718.02   509.5  718.66   525.4  717.23   553.3  716.76   569.2  715.27
#Mann= 7 ,-1 , 0
       0     .06       0   15.67     .12       0  184.68    .045       0
  199.75     .12       0   253.3     .06       0   400.5    .016       0
  451.81     .12       0
Bank Sta=184.68,199.75
XS Rating Curve= 0 ,0
Exp/Cntr=0.3,0.1

Type RM Length L Ch R = 1 ,11966.3 ,310,320.3,314.9
XS GIS Cut Line= 2
     2359225.267      311442.798     2359252.828      310852.412
#Sta/Elev= 30
       0  708.06   38.48705.2059    87.9  702.95   103.8  701.52   115.8  701.73
   123.8  701.25   147.8  700.94   171.7  701.44   215.6  700.43   223.6  699.74
   230.1  698.12   235.6  697.15   245.1  697.95   247.6  698.62   255.6  702.45
   259.6   703.7   271.6  705.22   279.5  705.87   327.8707.7507   355.4  709.76
  408.38712.1667   423.3   712.7  437.95712.4885   447.3  713.04   459.2  712.98
  468.24 714.985   495.2  715.53   531.1  715.46   555.1   714.5     591  714.73
#Mann= 8 ,-1 , 0
       0     .06       0   38.48     .12       0   230.1    .045       0
   245.1     .12       0   327.8     .06       0  408.38     .12       0
  437.95    .016       0  468.24     .12       0
Bank Sta=230.1,245.1
XS Rating Curve= 0 ,0
Exp/Cntr=0.3,0.1

Type RM Length L Ch R = 1 ,11646   ,213.3,215,217.2
XS GIS Cut Line= 2
     2359429.694      311481.861     2359600.267      310958.423
#Sta/Elev= 30
       0  707.85   61.64 703.755   111.7  701.65   123.7   700.6   147.6  700.99
   167.6  699.72   179.5  698.32   195.5  698.98   203.5  697.96   215.4  696.96
  218.39697.9717   223.4  699.49   227.4  699.77   235.4  699.84   247.3  699.02
   279.2  701.14   307.2  703.56   319.2  705.69   347.1  706.69  352.45706.0177
     359  704.64     367  704.99     379  704.42  388.84705.7518   394.9  706.11
   418.9  705.55   438.8  705.73  491.34707.0652  532.66707.7621   550.5   708.6
#Mann= 8 ,-1 , 0
       0     .06       0   61.64     .12       0   203.5    .045       0
  218.39     .12       0  352.45    .016       0  388.84     .06       0
  491.34     .12       0  532.66     .06       0
Bank Sta=203.5,218.39
XS Rating Curve= 0 ,0
Exp/Cntr=0.3,0.1

Type RM Length L Ch R = 1 ,11431   ,244.6,247.4,246
XS GIS Cut Line= 2
     2359603.088      311565.303     2359810.337       311053.15
#Sta/Elev= 30
       0  706.14   36.75703.8672    39.8  703.73    51.7  702.28    67.6  701.22
   111.3   699.5   135.1  699.08     155  699.25   166.9  698.31   174.9  698.02
   182.8   698.3     209698.1915   254.4   698.2   262.3  697.44   265.2  696.86
   270.3  696.03   274.3     696   280.2   696.7   290.2  698.31   298.1  698.78
     318  698.57   329.9  699.48   341.8  699.34  354.83700.1409  391.76700.8139
  404.78701.1776   433.2  702.06   457.1  703.34  487.01 704.048   552.5  705.47
#Mann= 9 ,-1 , 0
       0     .12       0   36.75     .06       0     209     .12       0
   265.2    .045       0   280.2     .12       0  354.83    .016       0
  391.76     .06       0  404.78     .08       0  487.01     .06       0
Bank Sta=265.2,280.2
XS Rating Curve= 0 ,0
Exp/Cntr=0.3,0.1

Type RM Length L Ch R = 1 ,11183.6 ,131,130.8,131.2
XS GIS Cut Line= 2
     2359752.051      311671.584     2360035.723      311155.203
#Sta/Elev= 30
       0  705.18   29.01705.4084      63 704.355   77.07703.7049   123.4  702.73
   141.3  703.74  145.17703.4878   179.1  702.16   213.1702.3262  230.14702.6253
   258.8  700.71  275.59697.2222   290.6  696.25   298.6  695.84   306.5  696.21
   322.4  698.64   334.4  697.63   346.3  698.22  369.59697.7092  371.25697.6554
   382.2  697.57   394.1  699.88     414  701.02     422  700.74   429.9  699.07
  435.81698.7773  437.96698.8382   481.7  699.51  568.48703.5998   589.2  705.52
#Mann= 16 ,-1 , 0
       0     .06       0   29.01     .12       0      63     .08       0
   77.07     .12       0   141.3     .08       0  145.17     .12       0
   213.1     .08       0  230.14     .12       0  275.59     .07       0
   290.6    .045       0   306.5     .07       0  369.59     .12       0
  371.25    .016       0  435.81     .12       0  437.96     .06       0
  568.48     .08       0
#XS Ineff= 2 , 0
          279.88  700.28  320.74          700.26
Permanent Ineff=
       F       F
Bank Sta=290.6,306.5
XS Rating Curve= 0 ,0
Exp/Cntr=0.3,0.1

Type RM Length L Ch R = 1 ,11052.9 ,154.9,181.1,190.3
XS GIS Cut Line= 2
     2359872.494      311718.241     2360156.165      311201.861
#Sta/Elev= 30
       0  702.15   13.33 701.735    35.8  701.97   51.04702.5606    71.7  703.44
    87.6   703.4   111.5  702.55  186.99  701.64  212.71702.2057     219  701.93
   222.9   701.1   230.9  698.42   234.9  698.13   242.8  699.25   246.8  698.98
   258.8  696.84   270.7  696.44   278.7   695.7   282.6  695.57   294.6   695.7
   326.4  696.88   358.3  696.95   394.1  698.75  407.28698.6128  458.91699.4833
   473.7  699.55  490.49700.6289   501.6  700.27   513.5   701.3   589.2  703.99
#Mann= 10 ,-1 , 0
       0     .12       0   13.33     .06       0   51.04     .08       0
  186.99     .06       0  212.71     .12       0   278.7    .045       0
   294.6     .12       0  407.28     .06       0  458.91     .08       0
  490.49     .06       0
#XS Ineff= 2 , 0
          260.06  699.39  315.17          699.35
Permanent Ineff=
       F       F
Bank Sta=278.7,294.6
XS Rating Curve= 0 ,0
Exp/Cntr=0.3,0.1

Type RM Length L Ch R = 1 ,10871.7 ,249.8,259.3,268.4
XS GIS Cut Line= 3
     2359892.802      311713.957     2359965.502      311597.855
      2360487.42      311587.004
#Sta/Elev= 30
       0  701.49    36.7701.7377   48.14702.1426    58.7   702.9   84.02702.5433
  118.53 701.864  137.66701.5103   196.8  699.91   212.7  697.35   220.7  696.96
   230.6  694.24   240.6  693.42   245.6  694.52   252.6  695.65   260.5  695.67
   300.4   695.2   312.3   694.1   320.3  695.76  333.18696.2851   360.1  696.07
     384  697.08   455.8   698.2  491.84699.4062  521.36700.8444   579.3  703.34
   603.2  703.57   627.1   704.6  637.16704.2885   647.1  704.26     659  705.17
#Mann= 12 ,-1 , 0
       0     .06       0    36.7     .12       0   48.14     .08       0
   84.02     .06       0  118.53     .08       0  137.66     .12       0
   230.6    .045       0   245.6     .12       0  333.18     .06       0
  491.84     .08       0  521.36     .06       0  637.16     .12       0
Bank Sta=230.6,245.6
XS Rating Curve= 0 ,0
Exp/Cntr=0.3,0.1

Type RM Length L Ch R = 1 ,10612.4 ,165.5,156.1,146.4
XS GIS Cut Line= 3
     2359881.951      311741.084     2360154.304      311849.591
     2360424.486      311787.742
#Sta/Elev= 30
       0  701.37    11.9  700.52    35.7  696.25    47.5  695.02    63.4  694.74
    71.3  695.36    91.1  694.54   142.6  694.39   154.5  693.94  164.13694.1719
   186.2  694.56   194.1  694.28  199.83693.0676     202   692.5     206  692.23
   213.9  693.02   221.9  695.96   229.8  697.08   241.7  700.02   249.6  700.45
   257.5  701.76  283.81701.4722     313  702.17   415.9  708.37   447.6  709.68
   463.4  709.52   471.4  710.01   518.9  708.66   534.7  707.35   570.3   705.4
#Mann= 5 ,-1 , 0
       0     .06       0  164.13     .12       0  199.83    .045       0
   213.9     .12       0  283.81     .06       0
Bank Sta=199.83,213.9
XS Rating Curve= 0 ,0
Exp/Cntr=0.3,0.1

Type RM Length L Ch R = 1 ,10456.3 ,398.9,393.9,376.4
XS GIS Cut Line= 3
     2359744.147      312081.796     2359847.229      311929.886
      2360406.04      311902.759
#Sta/Elev= 30
       0  705.25    31.9  703.47    75.8  698.63  102.23697.1346   159.6  697.38
   171.6  695.93   179.6  696.85   199.6  696.23   207.6  696.77   243.5  693.84
   267.5  692.98   287.5  693.34   311.5  691.09   323.4  691.01   327.4   691.1
   339.4   693.2   355.4  694.36   375.4  698.86   411.4  700.59   415.4  700.44
   423.4  698.12   427.4  698.09   435.3   700.4   451.3  701.74  477.89700.9376
  557.31704.5635  615.34708.3467   687.1  712.63  718.46 713.362     743  714.15
#Mann= 8 ,-1 , 0
       0     .06       0  102.23     .12       0   311.5    .045       0
   327.4     .12       0  477.89     .06       0  557.31     .12       0
  615.34     .06       0  718.46     .08       0
Bank Sta=311.5,327.4
XS Rating Curve= 0 ,0
Exp/Cntr=0.3,0.1

Type RM Length L Ch R = 1 ,10062.3 ,517.6,526.3,519.5
XS GIS Cut Line= 2
     2359940.545      312347.638      2360406.04      311948.332
#Sta/Elev= 30
       0  708.64    31.9  705.48  104.32696.5285   127.4  695.48   143.4  693.13
   155.3  692.93  162.46  691.19   167.3  689.74   171.2  689.59   177.4 690.892
  189.07692.1621   203.1  692.74   250.9  692.06  280.32692.3648   294.7  691.39
   306.6  691.54   318.6  692.64   322.6  693.34   330.5  696.35   338.5  696.78
   346.5  698.49   370.4  700.45  401.73700.4247  407.77700.3286   469.9  705.95
   481.9  708.63   509.8  710.14  522.15712.0977  612.03714.2327   613.3  714.22
#Mann= 10 ,-1 , 0
       0     .06       0  104.32     .12       0  162.46    .045       0
   177.4     .12       0  189.07     .06       0  280.32     .12       0
  401.73     .06       0  407.77     .12       0  522.15     .06       0
  612.03     .08       0
Bank Sta=162.46,177.4
XS Rating Curve= 0 ,0
Exp/Cntr=0.3,0.1

Type RM Length L Ch R = 1 ,9536.1  ,292.8,295.4,298.1
XS GIS Cut Line= 3
     2360257.385      312597.204     2360536.248      312278.193
     2360523.227      312079.626
#Sta/Elev= 30
       0  702.66      52   698.3   79.37697.1279    95.9  696.36   119.9  696.15
   147.9  694.68   163.9  694.72   167.9  694.06   175.9   691.6   187.9  690.17
   223.8   690.8   263.8  690.74   279.8  689.82   289.8  687.84   295.8   687.5
   304.8  688.06   315.8   689.8   335.8   691.2  360.61 695.636   363.8  696.29
   399.7  697.59   423.7   697.2   431.7  697.79   447.6   697.6   463.5   698.2
     563  708.68   578.9  710.03  598.73710.6274  600.41710.6863   622.7  711.62
#Mann= 7 ,-1 , 0
       0     .06       0   79.37     .12       0   289.8    .045       0
   304.8     .12       0  360.61     .06       0  598.73     .12       0
  600.41     .06       0
Bank Sta=289.8,304.8
XS Rating Curve= 0 ,0
Exp/Cntr=0.3,0.1

Type RM Length L Ch R = 1 ,9240.6  ,257,259,260.2
XS GIS Cut Line= 2
     2360461.378      312736.093       2360881.3      312381.275
#Sta/Elev= 30
       0  699.45       8  699.13    71.7  692.91    79.7  692.55    87.6  692.87
   98.61692.5049   119.5  692.71   139.4   691.8   155.4  689.12   167.3   688.9
   187.2  689.22   219.1  688.76   228.9  687.23     235  686.45     239  686.52
   243.9  687.61     247  688.56   258.9  689.09   274.9  688.97  291.99689.3765
   298.8  689.82   314.7  691.51   326.7  691.61   386.4  694.34   402.4  694.68
   430.2  695.82   454.2  695.85   466.1  696.19     478  696.01   549.8  697.23
#Mann= 5 ,-1 , 0
       0     .06       0   98.61     .12       0   228.9    .045       0
   243.9     .12       0  291.99     .06       0
Bank Sta=228.9,243.9
XS Rating Curve= 0 ,0
Exp/Cntr=0.3,0.1

Type RM Length L Ch R = 1 ,8981.6  ,309.3,322.8,330.4
XS GIS Cut Line= 3
     2360542.759      312868.471      2360648.01      312870.641
      2361035.38      312576.588
#Sta/Elev= 30
       0  706.47   12.54703.8405    50.7  695.09      78   691.4   105.3  690.28
   117.2  690.77   133.2   690.6   141.2   689.4   153.1  686.24   157.1  685.65
     173  687.24     201  687.52   208.9  687.24   216.9   685.6   220.9  685.33
   232.8  685.77   240.8  686.59   248.8  685.21   256.8  684.22  263.67685.1754
   272.7  687.47  288.48688.5671   304.6  690.13   316.6  692.16   328.5  693.53
   348.4  694.92   392.3  695.22   436.1  694.74   511.9   695.5   591.6  698.48
#Mann= 5 ,-1 , 0
       0     .06       0   12.54     .12       0   248.8    .045       0
  263.67     .12       0  288.48     .06       0
Bank Sta=248.8,263.67
XS Rating Curve= 0 ,0
Exp/Cntr=0.3,0.1

Type RM Length L Ch R = 1 ,8658.8  ,371.9,354.6,336.7
XS GIS Cut Line= 4
     2360540.588       313088.74     2360654.521      312994.339
     2360831.387      312986.744     2361109.165      312756.709
#Sta/Elev= 30
       0  713.01      32  708.19      40  706.32      48  703.61      72  698.94
      80  696.63      88  695.08      96  694.53     120  691.39   175.5  688.39
   179.4  687.67  190.07 683.592   199.1  682.67  204.98683.5098   214.8  684.29
   226.6  686.74   238.4  688.46   254.2  687.57   273.8  687.36   305.3  688.28
     329  689.88   352.7  692.61  365.44693.0579   388.4  693.37   400.3   694.3
   416.2  694.69   455.8  694.33   479.6  694.94   566.8   695.2   685.6  697.14
#Mann= 4 ,-1 , 0
       0     .12       0  190.07    .045       0  204.98     .12       0
  365.44     .06       0
#XS Ineff= 2 , 0
                          294.74           689.4
Permanent Ineff=
       F       F
Bank Sta=190.07,204.98
XS Rating Curve= 0 ,0
Exp/Cntr=0.3,0.1

Type RM Length L Ch R = 1 ,8304.2  ,362.5,370.9,388.4
XS GIS Cut Line= 2
      2360718.54      313356.752     2361159.078      312907.534
#Sta/Elev= 30
       0  715.51    27.9   713.5    47.8  711.21    55.8  710.16    87.6  703.89
   115.5  699.62   191.1  690.28  206.97689.0856     235  687.48   246.9  685.39
   254.9  684.83   278.8  685.31   294.7  686.71   306.6  686.12   314.6  686.53
   334.5   685.1   346.4  683.14   362.4  682.88   374.3  681.32   378.3   681.7
  380.89682.9756   385.7685.5577   390.2  687.24   398.2  688.42   406.2   689.1
   418.1  691.11     438  693.18   561.5  693.96   613.2  695.15   629.2  695.08
#Mann= 5 ,-1 , 0
       0     .06       0  206.97     .12       0   362.4    .045       0
  380.89     .12       0   385.7     .06       0
Bank Sta=362.4,380.89
XS Rating Curve= 0 ,0
Exp/Cntr=0.3,0.1

Type RM Length L Ch R = 1 ,7933.3  ,194.4,200.4,206.2
XS GIS Cut Line= 3
     2360758.687      313430.537     2361067.932      313329.626
     2361316.413      313069.209
#Sta/Elev= 30
       0  713.01    31.7  711.38     119  702.83   186.4  691.38   210.2  688.49
     234  687.58   285.6  687.82  304.81686.6404   333.3  685.53   341.3  685.76
   353.3  684.26   361.3   683.8   381.3  683.78   397.3  682.98   409.3  683.34
   421.3  681.98   433.3  681.54   442.1  679.94   453.3  679.44   457.1  679.65
   477.3  683.52  479.93683.5989   481.3  683.64   485.3  685.49   489.3  686.38
   509.3  687.94   517.3  689.38   529.3  690.03   605.2  693.18   685.2  693.88
#Mann= 5 ,-1 , 0
       0     .06       0  304.81     .12       0   442.1    .045       0
   457.1     .12       0  479.93     .06       0
Bank Sta=442.1,457.1
XS Rating Curve= 0 ,0
Exp/Cntr=0.3,0.1

Type RM Length L Ch R = 1 ,7732.9  ,194.2,190.2,183.3
XS GIS Cut Line= 3
     2360814.026      313501.067     2361123.271      313488.046
     2361474.833      313263.436
#Sta/Elev= 30
       0  707.12   103.2  701.08     123  699.53   190.5  692.95   222.2  690.75
   273.8  688.78   313.5  684.92   349.2  684.32  355.65683.6015   361.2  683.05
   377.1  683.42   396.9  682.97   404.9  681.24   412.8  681.76   432.3  678.29
   436.7  678.02   447.3  678.09   460.5  680.71   484.3  682.09   504.2  684.29
   508.2  684.93   520.1   688.8   543.9  689.38  570.02 689.191   611.5  689.84
   639.3  690.81   667.1  693.04   694.9  693.83  713.97 695.337   726.7   696.2
#Mann= 6 ,-1 , 0
       0     .06       0  355.65     .12       0   432.3    .045       0
   447.3     .12       0  570.02     .06       0  713.97     .12       0
#XS Ineff= 2 , 0
           380.6   684.4
Permanent Ineff=
       F       F
Bank Sta=432.3,447.3
XS Rating Curve= 0 ,0
Exp/Cntr=0.3,0.1

Type RM Length L Ch R = 1 ,7542.7  ,188.9,179.9,184.2
XS GIS Cut Line= 2
     2361128.696      313816.822      2361499.79      313333.966
#Sta/Elev= 30
       0  694.77   94.13691.5327  113.06690.0361   123.4  689.25   155.2  685.38
   172.7683.6977     199  681.86   230.9  681.81   270.7  681.01   274.6  680.76
   282.6  679.26   298.5  678.64   302.5   677.9   310.5  677.02   318.4  677.87
   334.3  680.86   350.3  687.54   354.2  688.72   358.2  689.08   378.1  688.43
     406  689.07   441.8  689.19   509.5  688.59   537.3   689.8   549.3  691.27
   561.2  693.54   569.2  693.82  581.71695.1996  598.94695.9203     609  696.69
#Mann= 8 ,-1 , 0
       0     .06       0   94.13     .12       0  113.06     .06       0
   172.7     .12       0   302.5    .045       0   318.4     .12       0
  581.71     .06       0  598.94     .12       0
Bank Sta=302.5,318.4
XS Rating Curve= 0 ,0
Exp/Cntr=0.3,0.1

Type RM Length L Ch R = 1 ,7362.8  ,101.4,94,87.6
XS GIS Cut Line= 3
     2361368.496      313932.924     2361461.812      313528.193
     2361560.554      313356.752
#Sta/Elev= 30
       0  692.91      20  691.32  114.24687.5397   131.8  686.82   155.8  683.55
   187.7  680.73   195.7  680.43   207.7  680.63   215.7   679.3   219.7  679.24
   227.6  679.95   243.6   680.5   247.6  679.88   251.6  678.47   259.6677.6263
   267.6  677.46   275.6   677.8   287.6   678.8   295.5  680.38   327.5  681.91
   371.4  686.08   415.4   687.4   458.9  686.32   474.7   686.3   514.3   687.6
   522.2  688.61   534.1  692.85   545.9  693.06   557.8  694.02   613.2  696.92
#Mann= 4 ,-1 , 0
       0     .06       0  114.24     .12       0   259.6    .045       0
   275.6     .12       0
Bank Sta=259.6,275.6
XS Rating Curve= 0 ,0
Exp/Cntr=0.3,0.1

Type RM Length L Ch R = 1 ,7268.9  ,102.9,106.4,109.4
XS GIS Cut Line= 4
     2361445.536      313958.966     2361517.151       313865.65
     2361516.066      313457.664     2361567.064      313364.348
#Sta/Elev= 30
       0  691.17    39.2  689.06   95.19684.8235   105.9  683.32   121.6   682.1
   161.6  680.08  186.21 679.767  279.42679.8209   293.6  679.76  302.67678.2679
  306.48677.3438   313.6   676.7   321.6  676.87  323.47677.3001   334.8 680.376
   341.6  681.31   373.6  683.21   385.6  684.62   409.6  685.57   457.6  686.63
   493.6  686.33   529.6  686.92   537.4  687.52   541.4  688.37   553.2   693.1
     565  693.14   576.8  694.03   600.4  694.79   612.3  695.89     632   696.5
#Mann= 8 ,-1 , 0
       0     .06       0   95.19     .12       0  186.21     .06       0
  279.42     .12       0  302.67     .06       0  306.48    .045       0
  323.47     .06       0   334.8     .12       0
#XS Ineff= 2 , 0
          144.48  683.02
Permanent Ineff=
       F       F
Bank Sta=306.48,323.47
XS Rating Curve= 0 ,0
Exp/Cntr=0.3,0.1
